--- BIGRUN2.prj (project) ---

Proj Title=BIGRUN2
Current Plan=p01
Default Exp/Contr=0,0
English Units
Geom File=g01
Flow File=f01
Plan File=p01
BEGIN DESCRIPTION:
END DESCRIPTION:
DSS Export Rating Curves= 0
DSS Export Rating Curve Sorted= 0
DSS Export Volume Flow Curves= 0
DXF OffsetX= 0
DXF OffsetY= 0
DXF ScaleX= 0
DXF ScaleY= 0

--- BIGRUN2.p01 (plan) ---

Plan Title=Floodplain
Program Version=4.00
Geom File=g01
Flow File=f01
K Sum by GR=0
Std Step Tol=0.01
Critical Tol=0.01
Num of Std Step Trials=20
Max Error Tol=0.3
Flow Tol Ratio=0.001
Split Flow NTrial=30
Split Flow Tol=0.02
Split Flow Ratio=0.02
Log Output Level=0
Friction Slope Method=1
Unsteady Friction Slope Method=2
Unsteady Bridges Friction Slope Method=1
Global Log Level=0
CheckData=False
Run HTab=0
Run UNet=0
Run PostProcess=0
UNET Theta=0
UNET Theta Warmup=0
UNET ZTol=0
UNET ZSATol=0
UNET MxIter=0
UNET MaxInSteps=0
UNET DtIC=0
UNET DtMin=0
UNET MaxCRTS=0
UNET WFStab=0
UNET SFStab=0
UNET WFX=0
UNET SFX=0
UNET DSS MLevel=0
UNET DZMax Abort=0
UNET Convert EG Bridges=0
UNET Use Existing IB Tables=0
UNET Froude Limit=0
UNET Froude Power=0
Write IC File=0
Echo Input=False
Echo Output=False
Write Detailed=0

--- BIGRUN2.f01 (steady flow) ---

Flow Title=NFF Regression Equation
Program Version=5.03
Number of Profiles= 1
Profile Names=P100yr
River Rch & RM=BIGRUN2,Main            ,13168.1
512.1093
River Rch & RM=BIGRUN2,Main            ,12613.1
 543.886
River Rch & RM=BIGRUN2,Main            ,11469.7
581.5239
River Rch & RM=BIGRUN2,Main            ,10682.9
641.1736
River Rch & RM=BIGRUN2,Main            ,7707.5
707.0119
River Rch & RM=BIGRUN2,Main            ,7363.8
800.7233
River Rch & RM=BIGRUN2,Main            ,5599
821.9627
River Rch & RM=BIGRUN2,Main            ,3786.7
910.9582
River Rch & RM=BIGRUN2,Main            ,196.1
1012.129
Boundary for River Rch & Prof#=BIGRUN2,Main            , 1
Up Type= 0
Dn Type= 3
Dn Slope=0.00987
DSS Import GetInterval= 0
DSS Import GetPeak= 0
DSS Import FillOption= 0

--- BIGRUN2.g01 (geometry) ---

Geom Title=USGS 10m DEM
Program Version=4.10

River Reach=BIGRUN2         ,Main
Reach XY= 30
     2370018.671       419040.25     2370254.782      419298.931
      2370509.99      419193.028     2370652.351      419286.778
     2370682.834      419625.218     2370857.212      419753.792
     2371292.976      419569.764     2371607.212      419708.653
     2372027.669      419475.262     2372707.907      419574.972
      2372947.49      419451.708     2373074.226      419210.389
     2373227.105      419150.305     2373380.968      418780.108
     2373589.952      418740.236     2373895.407      418357.959
      2374501.31      418291.986     2374909.296      418033.306
     2375074.226      417658.306     2375218.323       417665.25
      2375345.06      417408.306     2375973.532      416949.972
     2376777.351      416646.153     2376952.698      416830.181
     2377246.101      416719.069      2377478.74       416781.57
     2377707.907      417623.583     2377725.268      418482.958
     2377865.227      418581.594     2378023.092      419237.038

Type RM Length L Ch R = 1 ,13168.1 ,313.4,300.8,280.2
XS GIS Cut Line= 2
     2369897.214      419077.485     2370153.985      419018.241
#Sta/Elev= 30
       0  578.96    31.9  566.08    35.9  564.15    43.9  558.83    51.9  555.12
    71.9  544.87    83.8  539.34    95.8  534.26    99.8  532.77   107.8  530.24
   119.1  525.17   123.8  523.76   127.8  523.46   131.8  523.78   134.1  524.54
   135.8  525.11   139.7  526.84   143.7  527.65   159.7  527.12   171.7   526.2
   179.7  526.44   187.7  526.09   191.6   526.3   195.6  527.15   203.6  530.03
   207.6  531.84   215.6  535.97   227.6  541.03   239.6  546.48   263.5  556.91
#Mann= 3 ,-1 , 0
       0     .12       0   119.1    .045       0   134.1     .12       0
Bank Sta=119.1,134.1
XS Rating Curve= 0 ,0
Exp/Cntr=0.3,0.1

Type RM Length L Ch R = 1 ,12867.3 ,267.6,254.2,230.4
XS GIS Cut Line= 4
      2370146.39       419379.57     2370154.367      419307.605
     2370212.336      419193.383     2370236.451      419092.026
#Sta/Elev= 30
       0  545.41    11.4  542.16    30.5  535.31    38.1  533.01    49.5  530.02
    57.2  528.61    64.8  526.73    68.6  526.02      84  524.79    95.7  525.34
   122.9   525.2   146.2  523.59     150  522.87   153.9  521.76   157.8  520.96
   161.7  521.13   165.6  522.66   169.4  524.44   173.3  525.23   188.8  527.43
   192.7  527.64   208.2  529.18   215.9  530.54   223.6  532.42   239.1  537.29
   246.8  540.21   258.4  545.25   277.7  554.37   293.1  560.72   304.7  564.77
#Mann= 3 ,-1 , 0
       0     .12       0     150    .045       0   165.6     .12       0
#XS Ineff= 2 , 0
          107.28  525.74
Permanent Ineff=
       F       F
Bank Sta=150,165.6
XS Rating Curve= 0 ,0
Exp/Cntr=0.3,0.1

Type RM Length L Ch R = 1 ,12613.1 ,264.5,267.6,269.7
XS GIS Cut Line= 3
     2370436.103       419379.57     2370398.126       419315.55
     2370378.595      419094.196
#Sta/Elev= 30
       0  545.65     7.8  544.51    15.7   542.3    39.2  534.34    66.6     527
    70.5  526.32    86.3  526.04    98.2  523.98   114.1   524.6     126  524.39
     130  523.63     134  521.77   137.9  518.56   141.9  516.82   145.9   516.8
   149.8  517.16   153.8  518.41   157.8  519.18   165.7  519.48   173.6  520.99
   177.6  521.38   213.3  523.45   221.3  524.59   229.2  526.55   241.1  531.41
     249  535.23   272.8  548.89   280.8  553.03   288.7  557.75   296.6  561.69
#Mann= 3 ,-1 , 0
       0     .12       0   137.9    .045       0   153.8     .12       0
#XS Ineff= 2 , 0
                          181.42          522.26
Permanent Ineff=
       F       F
Bank Sta=137.9,153.8
XS Rating Curve= 0 ,0
Exp/Cntr=0.3,0.1

Type RM Length L Ch R = 1 ,12345.5 ,204.8,229.1,253
XS GIS Cut Line= 3
     2370532.675      419391.505     2370588.013      419301.445
     2370595.609      419099.622
#Sta/Elev= 30
       0  543.36     7.8  540.97    15.7  537.96    31.3     531    43.1  526.13
    54.8  521.73    58.7  520.67    74.4  518.65    78.3  517.81    86.1  518.15
      94  519.01   105.7  518.34   113.6  518.69   117.6  518.52   121.5  517.63
  127.69515.5399   133.4  514.77   137.4  514.76  143.14515.6201   149.3  516.77
   165.1  518.08     181   518.6   188.9  520.09   200.8  521.24   236.4  523.28
     280  527.42   283.9  528.22   287.9  529.54   299.8  534.19   307.7  536.64
#Mann= 3 ,-1 , 0
       0     .12       0  127.69    .045       0  143.14     .12       0
#XS Ineff= 2 , 0
           94.63   519.4
Permanent Ineff=
       F       F
Bank Sta=127.69,143.14
XS Rating Curve= 0 ,0
Exp/Cntr=0.3,0.1

Type RM Length L Ch R = 1 ,12116.4 ,195.2,204,211.2
XS GIS Cut Line= 4
     2370572.822      419446.844     2370674.819      419440.333
      2370769.22      419395.846     2370880.805      419387.444
#Sta/Elev= 30
       0  541.88    15.7  538.71    31.4  534.51    39.3  531.65    51.1  526.57
    62.9  520.83    74.7  516.86    90.4  514.48   113.8  513.65   129.3  512.19
  135.68 509.588   140.9  508.42   149.5  509.63   156.3  512.19     164  512.78
   191.1  512.69   202.7  512.15   222.6  513.22   226.6   512.9   234.5  511.13
   242.5  510.74   246.5  512.44   250.5  516.06   258.5  524.17   262.5  527.68
   266.5  530.64   278.5  538.33   286.5  543.01   298.5  550.82   318.5  562.74
#Mann= 3 ,-1 , 0
       0     .12       0  135.68    .045       0   149.5     .12       0
Bank Sta=135.68,149.5
XS Rating Curve= 0 ,0
Exp/Cntr=0.3,0.1

Type RM Length L Ch R = 1 ,11912.4 ,190.4,169.8,148.5
XS GIS Cut Line= 3
     2370577.379      419617.851     2370801.338      419591.809
     2370892.484      419528.007
#Sta/Elev= 30
       0  545.24    31.6  535.85    43.5  532.86    47.5   531.1    51.4  528.82
    55.4   526.1    63.3  521.62    75.2  515.92      87  511.09    94.9  509.09
  100.73505.9922   102.8  504.92   106.8   504.5   110.8  504.79   118.7  505.91
   130.5  508.39   134.5  508.59   150.3   508.5   166.1  507.78     178  507.64
   189.9  506.96   197.8  507.03   201.7   507.8   217.6  512.67   221.5  513.54
   229.4   514.3   253.3  523.15   273.2  531.24   308.9  540.82   336.7  550.49
#Mann= 3 ,-1 , 0
       0     .12       0  100.73    .045       0   118.7     .12       0
Bank Sta=100.73,118.7
XS Rating Curve= 0 ,0
Exp/Cntr=0.3,0.1

Type RM Length L Ch R = 1 ,11742.7 ,297.6,273,244.1
XS GIS Cut Line= 3
     2370632.501      419816.853     2370734.497      419810.342
     2370894.003       419535.82
#Sta/Elev= 30
       0   544.2    27.5  536.58    39.3  532.43    51.1  527.01    66.8  519.02
    74.7  515.89    94.3  511.92     122  507.37   137.9  505.88   169.7  505.28
   177.6  505.49   193.5  504.32   209.4   504.7   225.2  503.62  233.93502.3879
   241.1  501.73     249  502.36     257  505.02   268.9  505.42   272.9  506.14
   280.8  509.35   284.8  509.81   312.6  510.99   316.5  511.88   332.4  517.01
   352.2   525.2   372.1  532.33     380  535.52   399.9  542.38   419.7  548.63
#Mann= 3 ,-1 , 0
       0     .12       0  233.93    .045       0     249     .12       0
Bank Sta=233.93,249
XS Rating Curve= 0 ,0
Exp/Cntr=0.3,0.1

Type RM Length L Ch R = 1 ,11469.7 ,227.5,233.6,239.4
XS GIS Cut Line= 3
     2371089.315       419854.83     2370973.213      419654.092
     2370964.532      419552.096
#Sta/Elev= 30
       0  552.91       8  548.94      16  545.44      40  532.92      48  528.54
      64  518.49      72  514.04      76  512.08      92  505.83     104  502.65
     120  499.11   123.9  498.69   131.9  499.84   135.9  499.72   143.3  498.22
   151.9  497.24   155.9  497.51   158.3  498.21   163.9  499.91   199.9  500.73
   203.9  501.26   215.9  504.15   223.9  505.11   235.8  505.86   243.7  507.32
   251.6  509.86   259.5  513.18     287  527.16   322.4  544.15   334.3  548.98
#Mann= 3 ,-1 , 0
       0     .12       0   143.3    .045       0   158.3     .12       0
Bank Sta=143.3,158.3
XS Rating Curve= 0 ,0
Exp/Cntr=0.3,0.1

Type RM Length L Ch R = 1 ,11236.1 ,261.1,286.7,311.9
XS GIS Cut Line= 3
     2371218.438      419801.662     2371234.714      419679.049
     2371192.397      419522.799
#Sta/Elev= 30
       0  534.93      20  526.72    35.9  519.94    47.9   515.4    67.8  508.42
    87.8  502.59    99.8  500.08   119.7  497.64   131.6  496.81   147.4  496.29
   151.3  495.31   155.3  494.02   159.2  493.36   171.1  494.28     179  496.19
   206.6   495.8   210.6  496.01   214.5   497.2   218.4  499.48   222.4  502.31
   230.3  508.55   234.2  511.89   242.1   517.5     250  523.98     254  527.03
   257.9  529.82   261.9  532.33   273.7  540.47   281.6  546.27   285.6  548.98
#Mann= 3 ,-1 , 0
       0     .12       0   155.3    .045       0   171.1     .12       0
Bank Sta=155.3,171.1
XS Rating Curve= 0 ,0
Exp/Cntr=0.3,0.1

Type RM Length L Ch R = 1 ,10949.4 ,292.9,266.5,239.9
XS GIS Cut Line= 3
      2371317.18       419775.62     2371498.386      419599.839
      2371482.11      419475.056
#Sta/Elev= 30
       0   518.5    15.8  515.22    31.6  512.66    51.3  510.64      71  506.73
    82.8  505.28    86.8  503.31    90.7   500.4    94.7  498.26    98.6  497.05
   110.4  494.55   130.2  492.37   138.1  491.07   153.8  491.45   173.6  490.15
  180.21 488.416   189.3     488  194.24 488.402   205.1  491.71   220.9  492.77
   252.5  493.53     280  494.97   299.6  496.77   303.6  497.76   323.2  504.41
   331.1  507.68   350.8  517.89   362.6  524.88   370.4  528.41   378.3  532.96
#Mann= 3 ,-1 , 0
       0     .12       0  180.21    .045       0  194.24     .12       0
#XS Ineff= 2 , 0
          149.85  492.06
Permanent Ineff=
       F       F
Bank Sta=180.21,194.24
XS Rating Curve= 0 ,0
Exp/Cntr=0.3,0.1

Type RM Length L Ch R = 1 ,10682.9 ,207.8,209.6,210.8
XS GIS Cut Line= 3
     2371677.423      419796.236      2371704.55      419709.431
     2371611.234       419463.12
#Sta/Elev= 30
       0  516.23    15.8  513.55    23.7  511.57    35.6  509.39    39.5  508.44
    47.4  505.31    59.3   503.9      83     497      91  494.99  100.03490.8991
   106.9  487.79   114.9  485.93   118.9   484.5   122.9  483.02   126.9  482.81
   130.8  483.43   133.2 484.468   138.8  486.16   142.8  486.56   158.8   486.1
   178.7  487.04   186.7  486.88   222.6  488.48   274.5  489.54   286.5  490.42
   290.5  491.36   298.5  494.25   310.4  500.11   326.4   509.2   354.3  526.45
#Mann= 4 ,-1 , 0
       0     .06       0  100.03     .12       0   118.9    .045       0
   133.2     .12       0
#XS Ineff= 2 , 0
                          192.78          487.94
Permanent Ineff=
       F       F
Bank Sta=118.9,133.2
XS Rating Curve= 0 ,0
Exp/Cntr=0.3,0.1

Type RM Length L Ch R = 1 ,10473.3 ,227,233.9,236.2
XS GIS Cut Line= 3
     2371885.756       419773.45     2371913.968      419693.155
     2371824.992      419404.526
#Sta/Elev= 30
       0  499.35    15.5   495.8    23.2  493.52    34.8  491.66    46.4  487.74
      58  485.89    73.5  485.56     105  484.04   112.9   484.3   128.8  483.78
   152.7  484.15   164.6  483.17   172.5  481.64   184.5  481.15     187481.6308
   192.4  483.19   196.4  483.63   212.3  483.55   224.2     483   232.2  482.15
   244.1  483.85     260  484.63   271.9  484.46   295.7  486.16   319.6   488.5
   327.5  490.12   335.5  491.13   355.4  496.22   371.2  500.83   387.1  504.56
#Mann= 3 ,-1 , 0
       0     .12       0   172.5    .045       0     187     .12       0
#XS Ineff= 2 , 0
                          260.47          485.07
Permanent Ineff=
       F       F
Bank Sta=172.5,187
XS Rating Curve= 0 ,0
Exp/Cntr=0.3,0.1

Type RM Length L Ch R = 1 ,10239.4 ,160.7,163.5,165
XS GIS Cut Line= 3
     2372076.077      419747.799     2372018.786      419433.997
     2372020.088      419359.778
#Sta/Elev= 30
       0  496.25      12  492.24      16  491.69    23.9  491.64    31.9  490.45
    35.9  489.34    39.9  486.43    43.9  482.28    47.8  479.56    59.8  479.46
    71.8  480.84   119.6  480.84   143.6  481.94   163.5  481.87   175.4  482.56
   227.3  481.04   247.2  479.88   259.2   480.5   267.2  478.14   275.1  477.16
   279.1  477.44  280.43478.0851   283.1  479.38   287.1   482.9   291.1  484.12
     303  485.41   342.4  487.59   358.1     490   369.8  494.23   393.2  506.43
#Mann= 3 ,-1 , 0
       0     .12       0   267.2    .045       0  280.43     .12       0
Bank Sta=267.2,280.43
XS Rating Curve= 0 ,0
Exp/Cntr=0.3,0.1

Type RM Length L Ch R = 1 ,10076   ,156.2,154,150.8
XS GIS Cut Line= 4
     2372196.086      419717.026     2372159.194      419574.882
     2372148.343      419472.886     2372192.831      419409.952
#Sta/Elev= 30
       0  495.89     7.9  492.95    19.8  487.61    27.8  486.41    31.8  485.51
    43.7  481.38    47.6  480.79    63.5  479.31    87.3  478.71   107.2  476.19
   115.1  478.26     123  479.09   170.5  479.26   178.4  478.67   185.6  476.15
   190.2  474.95   194.2  474.64   198.1  475.35   200.6  476.44     206  478.66
     210  479.01   221.8   479.3   233.6  478.48   237.6  478.78   245.5  479.92
   264.8  484.78   272.6  487.37   280.2  490.39   314.9  506.28   326.5  511.27
#Mann= 3 ,-1 , 0
       0     .12       0   185.6    .045       0   200.6     .12       0
Bank Sta=185.6,200.6
XS Rating Curve= 0 ,0
Exp/Cntr=0.3,0.1

Type RM Length L Ch R = 1 ,9922    ,69.7,88.2,107.6
XS GIS Cut Line= 3
     2372272.041       419702.92     2372305.678      419508.693
     2372278.551      419395.846
#Sta/Elev= 30
       0  503.39    27.6  492.22    39.4  486.28    43.4  484.58    47.3   483.8
    55.2   483.6    63.1  479.78      67  478.47      71  477.66    90.7  477.17
   114.3  477.24   130.1  476.66   145.9  477.07   177.4  476.96   189.2  477.37
     201  476.68   204.9  475.42   208.7  473.06   212.6  472.45   220.3  472.58
   222.4473.0646   224.2  473.48   231.9  476.57   235.8  477.45   239.7   479.4
   243.5  482.39   262.9   493.9   282.2  504.22   297.7  510.59   313.2  516.04
#Mann= 3 ,-1 , 0
       0     .12       0   208.7    .045       0   222.4     .12       0
Bank Sta=208.7,222.4
XS Rating Curve= 0 ,0
Exp/Cntr=0.3,0.1

Type RM Length L Ch R = 1 ,9833.8  ,94.1,93.2,92.5
XS GIS Cut Line= 4
     2372287.232      419712.686     2372316.529      419599.839
      2372417.44      419446.844      2372342.57      419382.825
#Sta/Elev= 30
       0  505.05    42.8  489.26    58.3  482.91    62.2  482.26      70  481.91
    77.7  480.22    81.6  479.79   116.6  477.06   144.5  476.98   172.4   475.3
   188.3  473.87   196.3  474.24   212.2  473.01   228.2  472.63   239.5  471.03
   244.1  470.01   248.1  470.03  253.54471.0311     260  472.74     268   476.1
     272  476.85  295.17478.6153  301.37478.9455   302.3479.0123   307.8  479.68
   311.7  480.63   323.5  484.94   343.2  493.26   370.8  502.09   398.4  507.87
#Mann= 6 ,-1 , 0
       0     .12       0   239.5    .045       0  253.54     .12       0
  295.17    .016       0  301.37     .06       0   302.3     .12       0
#XS Ineff= 2 , 0
           219.2   475.2
Permanent Ineff=
       F       F
Bank Sta=239.5,253.54
XS Rating Curve= 0 ,0
Exp/Cntr=0.3,0.1

Type RM Length L Ch R = 1 ,9740.6  ,96.7,90.2,83.3
XS GIS Cut Line= 4
     2372449.992      419710.516       2372413.1      419609.604
     2372514.011       419456.61     2372538.968      419371.974
#Sta/Elev= 30
       0   509.4       8  507.17    19.9  502.81    43.8  491.26    51.7  487.94
    55.7  485.96    59.7   483.5    63.7  481.95   89.38480.1261   107.4  479.71
  139.37477.8656   191.1  475.19     207  472.35     215  471.97     219  472.16
  224.26470.3137     227  469.43     231  469.22   238.9  469.64   242.9  470.39
   254.9  475.88   258.8  477.04   266.8  477.84   278.8  478.24   309.9  478.23
   313.7  478.14   325.2  476.94  332.34477.8213   340.6  478.76     379  480.48
#Mann= 6 ,-1 , 0
       0     .12       0   89.38    .016       0  139.37     .12       0
  224.26    .045       0   242.9     .12       0  332.34    .016       0
#XS Ineff= 2 , 0
          219.61  474.19
Permanent Ineff=
       F       F
Bank Sta=224.26,242.9
XS Rating Curve= 0 ,0
Exp/Cntr=0.3,0.1

Type RM Length L Ch R = 1 ,9650.3  ,244.6,228.2,211.4
XS GIS Cut Line= 4
     2372545.478      419701.835     2372540.053      419620.455
     2372598.647      419425.142     2372576.945      419363.294
#Sta/Elev= 30
       0  513.65     7.8  510.04    27.2  500.15      35  496.44    54.4  486.45
    62.1  481.88      66  479.93    81.6  473.64    89.6  472.83    97.6  472.72
   109.6  471.94   121.5  471.83   133.5  471.19   145.5  471.24   157.5  470.23
   161.5  469.42   169.5  468.83     177  469.54   181.5  470.77   189.5  471.45
   209.5  471.83   233.5  473.34   253.5  474.13   261.5   474.3   273.5  473.76
   293.2  474.81     297  475.15   308.6  477.26  325.54478.9964     351  480.22
#Mann= 4 ,-1 , 0
       0     .12       0   161.5    .045       0     177     .12       0
  325.54    .016       0
Bank Sta=161.5,177
XS Rating Curve= 0 ,0
Exp/Cntr=0.3,0.1

Type RM Length L Ch R = 1 ,9422.1  ,163.7,160.6,157.1
XS GIS Cut Line= 2
     2372807.848      419621.497      2372677.64      419322.017
#Sta/Elev= 30
       0  507.25    19.9  498.29    35.8   491.9    47.8  485.81    59.7  478.82
    63.7  475.97    71.7  469.01    74.8  467.13    75.7  466.58    79.6  465.79
    83.6  465.64    87.6  466.13    89.8   466.8    95.6   468.1   107.5  468.89
   115.5  468.74   123.5  469.27   171.2   468.9   187.2  469.66     231  470.32
   246.9  471.01   270.8  472.58   282.8  473.79   290.7  474.95   302.7  475.76
   306.6  476.76  308.71477.6937   310.6  478.53   318.6  479.92   326.6  480.42
#Mann= 4 ,-1 , 0
       0     .12       0    74.8    .045       0    89.8     .12       0
  308.71    .016       0
#XS Ineff= 2 , 0
                          190.35           470.3
Permanent Ineff=
       F       F
Bank Sta=74.8,89.8
XS Rating Curve= 0 ,0
Exp/Cntr=0.3,0.1

Type RM Length L Ch R = 1 ,9261.5  ,227.3,222.3,217.1
XS GIS Cut Line= 3
     2373013.143        419544.5     2372935.802      419510.258
     2372783.109      419268.892
#Sta/Elev= 30
       0  524.98     7.7  522.75    19.2  518.17    34.6  513.22    42.3  509.88
    88.6  484.96    96.5  480.15   112.4  467.69   116.3  465.89   119.4  465.18
   124.2  463.72   128.2  463.56   132.2  464.05   134.4  464.83   140.1  466.96
   144.1   467.3     152  466.86   171.8  466.84   183.8  467.53   191.7  467.32
   203.6  467.94   219.4     468   255.2  467.84   267.1  467.28   282.9  467.55
   326.6   470.9   346.4  473.87   351.2 475.491   362.3  478.45   370.2  479.09
#Mann= 4 ,-1 , 0
       0     .12       0   119.4    .045       0   134.4     .12       0
   351.2    .016       0
Bank Sta=119.4,134.4
XS Rating Curve= 0 ,0
Exp/Cntr=0.3,0.1

Type RM Length L Ch R = 1 ,9039.2  ,194.8,197.9,198.3
XS GIS Cut Line= 2
     2373122.952       419398.84     2372910.713      419185.299
#Sta/Elev= 30
       0   518.6     7.9  515.77    19.8  510.79    43.6   498.9    71.3  483.24
    83.2  476.94    95.1   469.2     103  464.98     107  463.84   110.9  463.65
   118.8  464.24   142.6  463.91   146.6  463.46   149.6  462.51   154.5   461.1
   158.5  460.65   164.6  462.24   170.3  464.02   174.3  464.32   190.2  464.33
     202  465.53     210  465.15   229.8  465.66   245.6  467.04  254.45468.3559
   261.5  469.07   281.3  470.07   289.2  473.59  294.75475.3294   301.1   477.1
#Mann= 5 ,-1 , 0
       0     .12       0   149.6    .045       0   164.6     .12       0
  254.45    .016       0  294.75     .12       0
#XS Ineff= 2 , 0
                          202.27          465.98
Permanent Ineff=
       F       F
Bank Sta=149.6,164.6
XS Rating Curve= 0 ,0
Exp/Cntr=0.3,0.1

Type RM Length L Ch R = 1 ,8841.3  ,72.4,65.4,60.1
XS GIS Cut Line= 3
     2373186.754      419324.231     2373179.159      419222.235
     2373026.164       419069.24
#Sta/Elev= 30
       0   508.4    15.7   503.6    23.6  501.85    35.4  498.76    55.1  491.28
    66.9  485.28    70.8  482.76    78.7  479.11    86.5  474.79    90.5  472.93
   106.2  464.51   114.1  461.63     118  459.79     122  458.49   125.9  458.64
   133.8  460.02   137.7  461.06   153.4  462.62   165.2  463.03  174.53 462.536
   188.8  462.61  214.43461.5663   243.9  463.72   251.8  464.53   263.6  467.32
   279.3  472.55   291.1  475.49     299  476.78   314.7  478.82   318.6  478.78
#Mann= 5 ,-1 , 0
       0     .12       0     118    .045       0   133.8     .12       0
  174.53    .016       0  214.43     .12       0
Bank Sta=118,133.8
XS Rating Curve= 0 ,0
Exp/Cntr=0.3,0.1

Type RM Length L Ch R = 1 ,8775.9  ,77.2,77.4,77.9
XS GIS Cut Line= 2
     2373339.749      419239.596     2373030.504      419054.049
#Sta/Elev= 30
       0  514.94    15.8  511.07    43.6  502.33    47.6   500.5    59.4  492.48
    67.4  489.75    75.3  487.94    87.2  482.34     103  478.75     107  477.28
   114.9  474.01   126.8  465.46   130.8  463.35   134.7  461.54   140.9 459.772
   146.6  458.28   150.6  457.97   154.6  458.54  156.43459.6085   162.5  462.37
  167.07462.2599   186.3  462.44  214.51460.9249   233.8  460.44   245.7  460.93
   281.4  464.38   289.3  465.82   309.1  471.56     321  474.13   360.6  478.31
#Mann= 5 ,-1 , 0
       0     .12       0   140.9    .045       0  156.43     .12       0
  167.07    .016       0  214.51     .12       0
Bank Sta=140.9,156.43
XS Rating Curve= 0 ,0
Exp/Cntr=0.3,0.1

Type RM Length L Ch R = 1 ,8698.5  ,143.9,149,153.4
XS GIS Cut Line= 3
      2373352.77      419209.214     2373284.538      419118.578
     2373073.907        418992.2
#Sta/Elev= 30
       0   514.2    11.7  509.81    23.5  504.68    31.3  502.09    62.6  485.24
      90  471.97    97.8  466.56  100.31465.1184   101.7  464.32   129.3   462.4
   137.2     461  142.25459.5773   145.1  458.43   149.1  457.44   153.1  457.19
     161  457.31     165  457.82   168.9  459.24   172.9  459.99   176.8  460.15
   220.4  458.95   252.1  460.18     264  461.14   295.7     465   303.6  465.72
   311.5  465.96   327.4  467.61   339.3   468.1   351.2  467.27   359.1  467.93
#Mann= 5 ,-1 , 0
       0     .12       0  100.31    .016       0  142.25     .12       0
   149.1    .045       0     165     .12       0
Bank Sta=149.1,165
XS Rating Curve= 0 ,0
Exp/Cntr=0.3,0.1

Type RM Length L Ch R = 1 ,8549.5  ,187.3,188.4,188.6
XS GIS Cut Line= 2
     2373438.491      419128.919     2373169.393      418881.523
#Sta/Elev= 30
       0  511.24    19.9  501.66    35.8  493.17    47.7  486.42   71.69474.2242
    79.5  467.83    83.4  465.13    95.4   464.6   103.3  463.72   107.3  462.43
   111.2  460.57   115.2  459.65   123.2  459.05  129.51459.0542  141.53459.1726
   162.9  458.31   202.6   458.4   222.5  458.54   238.4  458.23   254.3  456.46
   262.2  455.26   266.2   455.4   270.2  456.64   274.2  457.96   286.1  458.26
     290  458.74  308.34463.5249   313.9  464.83  357.49471.0365   365.5   472.3
#Mann= 9 ,-1 , 0
       0     .12       0   71.69    .016       0  129.51     .12       0
  141.53     .06       0   202.6     .12       0   254.3    .045       0
   270.2     .12       0  308.34     .06       0  357.49    .016       0
#XS Ineff= 2 , 0
          138.29  459.81
Permanent Ineff=
       F       F
Bank Sta=254.3,270.2
XS Rating Curve= 0 ,0
Exp/Cntr=0.3,0.1

Type RM Length L Ch R = 1 ,8361.1  ,262.6,271.2,274.3
XS GIS Cut Line= 2
     2373537.015      418978.267      2373309.15      418758.215
#Sta/Elev= 30
       0  488.62    19.8  474.82    23.8  472.35    31.7  468.79    35.6  466.57
   41.54462.6166    47.5  459.16    51.5  458.15    67.3   458.5    71.3  458.14
   80.37456.5039  102.68 455.388   134.6  454.78   150.5  455.43   166.3  455.13
   190.1  455.64   201.9  455.31  220.58455.7743   225.7   455.7  232.42453.9064
   233.6  453.52   237.6  453.31   249.5  453.92   265.3  455.99   269.3     457
   273.2  458.41   277.2   460.7   281.1  462.31  303.82466.4083   316.8  468.54
#Mann= 8 ,-1 , 0
       0     .12       0   41.54    .016       0   80.37     .12       0
  102.68     .06       0  220.58     .12       0  232.42    .045       0
   249.5     .12       0  303.82     .06       0
Bank Sta=232.42,249.5
XS Rating Curve= 0 ,0
Exp/Cntr=0.3,0.1

Type RM Length L Ch R = 1 ,8089.9  ,383.8,382.4,382.8
XS GIS Cut Line= 2
     2373719.306      418886.514     2373476.251      418584.865
#Sta/Elev= 30
       0  519.19      16  516.77    35.9  512.05    47.9  507.88    63.9  501.16
    79.9  493.65    87.9  489.21   107.8   476.5   111.8  472.52  116.58  465.82
   119.8  460.99   123.8  457.32   127.8  456.26   143.8  456.75   147.8  456.02
   155.8  453.13  171.97  452.22   187.7  451.91   195.5  450.27   203.7  449.55
   207.7  449.72   210.5  450.43   219.6  452.28   251.6  452.31   267.6  453.14
   295.5  453.48   303.5  454.03   315.5  455.91   355.4  463.91   387.4  469.13
#Mann= 5 ,-1 , 0
       0     .12       0  116.58    .016       0  171.97     .06       0
   195.5    .045       0   210.5     .06       0
#XS Ineff= 2 , 0
                          267.91          454.32
Permanent Ineff=
       F       F
Bank Sta=195.5,210.5
XS Rating Curve= 0 ,0
Exp/Cntr=0.3,0.1

Type RM Length L Ch R = 1 ,7707.5  ,328,343.7,358.9
XS GIS Cut Line= 2
     2373974.515      418712.252     2373717.353      418322.712
#Sta/Elev= 30
       0   515.3    39.9  501.34    63.8  491.48   103.7  473.59   123.7  466.34
   127.7  464.75  129.85463.2505   135.6  459.42   139.6  458.44   155.6  458.11
   167.6  454.27   176.4452.9145   227.4   448.2   247.4  447.51  275.09447.5858
   295.2  447.77   303.6  446.15   311.2  444.26   315.2   444.6   318.6   445.7
   323.2  447.31   327.1  447.61   343.1  447.19   351.1  447.92     363   451.9
     375  454.46     387  461.73   422.9  479.98   442.8  488.22   466.8  497.04
#Mann= 6 ,-1 , 0
       0     .12       0  129.85    .016       0   176.4     .06       0
  275.09     .12       0   303.6    .045       0   318.6     .12       0
Bank Sta=303.6,318.6
XS Rating Curve= 0 ,0
Exp/Cntr=0.3,0.1

Type RM Length L Ch R = 1 ,7363.8  ,257.6,249.5,240.6
XS GIS Cut Line= 3
     2374151.381      418585.299     2374081.937       418444.24
     2374112.319      418176.228
#Sta/Elev= 30
       0  531.05    19.6  522.97    70.8  499.24   129.7  468.91  136.08464.8266
   145.4   456.3   149.4   455.3   165.2   455.4   173.1  453.84  175.66452.4704
     185  447.53   200.9  443.89   216.7  443.65   232.6  441.98   237.5  440.96
   248.5  440.37  254.34440.9001   260.4  442.71   264.3  443.04   276.2  442.89
   292.1  444.62   311.9  445.72   315.9  446.18   323.8  448.66   327.8  450.38
   339.7   457.1   371.4  476.06   391.3  486.23   407.1  495.79     427  505.76
#Mann= 5 ,-1 , 0
       0     .12       0  136.08    .016       0  175.66     .12       0
   237.5    .045       0  254.34     .12       0
Bank Sta=237.5,254.34
XS Rating Curve= 0 ,0
Exp/Cntr=0.3,0.1

Type RM Length L Ch R = 1 ,7114.2  ,262.6,256.1,250
XS GIS Cut Line= 2
     2374374.905      418482.217      2374285.93      418156.696
#Sta/Elev= 30
       0  513.94    11.9  509.15    31.8  500.17    87.3   472.1   107.2  460.92
   112.6 455.419   115.1  452.31   119.1  448.76   123.1  447.97     139  447.96
   142.9  446.67  146.38444.8865   150.9   442.5   158.8  440.66   182.6  440.44
   190.6  438.62   198.5  438.09   206.4   438.3   218.4  441.06   234.2  442.88
   242.2   446.3   246.2  448.38   254.1  454.08     262  456.56     266  458.88
   273.9  466.15   285.8  473.96   309.7   487.1   329.5  499.58   337.5  504.08
#Mann= 5 ,-1 , 0
       0     .12       0   112.6    .016       0  146.38     .12       0
   190.6    .045       0   206.4     .12       0
Bank Sta=190.6,206.4
XS Rating Curve= 0 ,0
Exp/Cntr=0.3,0.1

Type RM Length L Ch R = 1 ,6858.1  ,318.6,316.2,313.5
XS GIS Cut Line= 3
     2374534.411      418447.495     2374584.324      418305.351
      2374450.86      418099.188
#Sta/Elev= 30
       0     504     7.9  501.21    23.8  494.33    35.7   488.3    55.5  479.32
    75.3  469.06    91.2  461.42     111   450.3   118.9  446.63   122.9  445.68
  137.35445.5097  169.09442.1628   206.1  440.44     214  438.12  219.63435.4427
     222   434.6   225.9  434.07   229.9  434.32   233.8  435.39   241.8  437.34
   285.3   437.3   289.3  437.76   293.3  438.91   301.2  443.05     317  452.63
   336.8  465.48   348.7  472.61   360.6  479.08   388.3  495.62   396.2  499.44
#Mann= 5 ,-1 , 0
       0     .12       0  137.35    .016       0  169.09     .12       0
  219.63    .045       0   233.8     .12       0
Bank Sta=219.63,233.8
XS Rating Curve= 0 ,0
Exp/Cntr=0.3,0.1

Type RM Length L Ch R = 1 ,6541.9  ,440.1,435.3,429.3
XS GIS Cut Line= 3
     2374888.143        418367.2     2374870.782      418164.292
     2374687.405      417924.491
#Sta/Elev= 30
       0  490.43    35.9  481.74    79.9   469.6   93.14465.3744   103.8  461.97
   119.8  454.86   127.8  452.97  141.01445.5515  144.36443.8112   147.8  442.59
   155.7  442.82   183.7  441.06  190.95438.1544   195.7   436.2   207.6  435.18
   223.5  434.73   235.4  435.04   275.2  433.83   287.1  430.97     295  430.08
   301.1  430.87   314.9  434.27   326.8  434.82   362.5  433.96   386.4  434.12
   410.2  435.14   430.1  437.32     446  441.36   473.8  451.13   505.5  459.81
#Mann= 7 ,-1 , 0
       0     .12       0   93.14     .06       0  141.01     .12       0
  144.36    .016       0  190.95     .12       0   287.1    .045       0
   301.1     .12       0
#XS Ineff= 2 , 0
          234.06  436.15
Permanent Ineff=
       F       F
Bank Sta=287.1,301.1
XS Rating Curve= 0 ,0
Exp/Cntr=0.3,0.1

Type RM Length L Ch R = 1 ,6106.6  ,521.2,507.6,526.4
XS GIS Cut Line= 2
     2375314.576      418038.424     2374925.036      417635.863
#Sta/Elev= 30
       0  482.11    43.7  467.41   91.02455.5016    99.3  450.88   119.2  450.07
  132.85446.7938   158.9  441.58   194.7  432.81   210.6  430.25   242.4   430.1
   250.3  429.62   301.9   429.9   313.9  429.67   325.8  428.21   333.7  429.52
   373.4  428.79  378.79427.9633   385.4  427.11   397.3  427.93   405.2  427.38
   425.1  428.61     445  428.66   448.9  429.36   460.8  434.19   464.8  435.21
   492.6  436.12   508.5  437.75   524.4  441.66   548.3  452.85   560.2  458.96
#Mann= 5 ,-1 , 0
       0     .12       0   91.02    .016       0  132.85     .12       0
  378.79    .045       0   397.3     .12       0
#XS Ineff= 2 , 0
          241.49  430.64
Permanent Ineff=
       F       F
Bank Sta=378.79,397.3
XS Rating Curve= 0 ,0
Exp/Cntr=0.3,0.1

Type RM Length L Ch R = 1 ,5599    ,478.3,496.4,497.2
XS GIS Cut Line= 2
     2375564.265      417778.145     2375135.539      417367.851
#Sta/Elev= 30
       0  474.95    35.8   464.1   62.52454.1961    67.7  451.94    71.7  449.11
    75.7  445.15    79.6  443.21    95.6  443.82    99.6  443.61  104.27442.1256
   111.5  439.04   115.5  438.05   155.3  429.69   215.1  423.76   266.8  423.59
   282.8   422.5   314.6  423.91   354.5  424.27   386.3   422.9   402.2   421.4
   410.2   420.7   418.2  421.51   426.2  422.65     450  423.39     462  429.78
   477.9  437.17   525.7  464.06   557.6  480.19   569.5  485.39   593.4  490.87
#Mann= 5 ,-1 , 0
       0     .12       0   62.52    .016       0  104.27     .12       0
   402.2    .045       0   418.2     .12       0
Bank Sta=402.2,418.2
XS Rating Curve= 0 ,0
Exp/Cntr=0.3,0.1

Type RM Length L Ch R = 1 ,5102.6  ,367.6,368.7,368.8
XS GIS Cut Line= 2
      2375846.26      417565.333     2375480.591      417124.795
#Sta/Elev= 30
       0  446.86       4   445.9   10.14443.1716    15.9   440.4    23.9  438.55
    39.8  435.25    51.7  433.88    71.6  433.17   103.4  430.49   143.1  428.81
   182.9  425.74   190.8   425.7   234.6  422.51   290.2  420.25   306.1  420.24
     334  419.35   365.8  417.75   378.1  416.47   385.7  416.12   393.1  416.58
   401.6  418.52   409.5  419.24   441.3  418.71   449.3   418.2   453.2   420.3
   461.2  428.49   465.2  431.38   473.1   436.1   528.8   461.1   572.5   477.3
#Mann= 4 ,-1 , 0
       0    .016       0   10.14     .12       0   378.1    .045       0
   393.1     .12       0
Bank Sta=378.1,393.1
XS Rating Curve= 0 ,0
Exp/Cntr=0.3,0.1

Type RM Length L Ch R = 1 ,4733.8  ,457.4,463.4,469.1
XS GIS Cut Line= 4
     2376096.911      417479.613     2376023.126      417278.875
     2375827.813      416988.077     2375628.161      417002.182
#Sta/Elev= 30
       0  441.58     7.9     442    15.8   441.5   24.75438.2646    31.7  435.91
    51.5  431.18    67.3  428.61      99  423.96   134.7   420.6   170.3  418.66
   257.7  417.37   321.4  417.34   361.2   415.4   432.8  416.27   440.8   415.5
   448.4  413.23   452.7  411.99   456.7  411.84   463.4  413.21   476.6  416.27
   524.4  416.21     572  418.57   579.9  419.51   630.9  428.54   642.7  429.63
   685.8  436.07   697.6  438.91   713.3  441.79   744.7  449.25   764.3  452.59
#Mann= 4 ,-1 , 0
       0    .016       0   24.75     .12       0   448.4    .045       0
   463.4     .12       0
#XS Ineff= 2 , 0
          340.14  417.69
Permanent Ineff=
       F       F
Bank Sta=448.4,463.4
XS Rating Curve= 0 ,0
Exp/Cntr=0.3,0.1

Type RM Length L Ch R = 1 ,4270.5  ,478.4,483.8,481.2
XS GIS Cut Line= 3
     2376400.156      417369.854     2376353.704      417097.339
     2376205.992      416713.721
#Sta/Elev= 30
       0  434.58   14.88433.4751    47.4  430.59   138.2  425.31  222.05417.8594
   248.8  416.34  350.39418.2732   364.2  418.76   376.2  416.47   388.2  417.65
   404.2  417.24   448.1  414.08     460  412.05     492  412.31   503.9  410.39
   515.9  410.53   523.9  411.92   547.8  413.05   563.8  411.99   567.8  410.72
   575.8  409.28   579.8  409.56   583.8  410.92   595.7  419.49   599.7  421.32
   607.7  423.34   627.6  427.27   655.6  430.82   667.6  431.37   687.5   433.9
#Mann= 6 ,-1 , 0
       0    .016       0   14.88     .12       0  222.05     .04       0
  350.39     .12       0   567.8    .045       0   583.8     .12       0
Bank Sta=567.8,583.8
XS Rating Curve= 0 ,0
Exp/Cntr=0.3,0.1

Type RM Length L Ch R = 1 ,3786.7  ,639.4,642,644
XS GIS Cut Line= 3
     2376689.359      417129.136     2376712.684       416951.88
     2376612.319      416533.432
#Sta/Elev= 30
       0  421.81     .65421.7726    39.7  419.82    63.6  417.56    83.4   416.3
   135.1  413.77   170.8  412.86   214.6  411.02   310.3  409.02   318.2  408.57
   330.2  407.02   338.2  407.89   354.1  408.68     370  408.18     390  409.26
   425.8  408.88   437.8  409.55   461.7  409.25   477.6  406.66   481.6  406.48
   493.6   406.8   497.5  408.76   505.5  415.18   509.5  417.33   517.5  420.13
   533.4  423.26   545.4  425.23   557.3  426.57   577.2  430.57   609.1  435.55
#Mann= 4 ,-1 , 0
       0     .06       0     .65     .12       0   477.6    .045       0
   493.6     .12       0
#XS Ineff= 2 , 0
          262.23  410.62
Permanent Ineff=
       F       F
Bank Sta=477.6,493.6
XS Rating Curve= 0 ,0
Exp/Cntr=0.3,0.1

Type RM Length L Ch R = 1 ,3144.8  ,451.1,486,510.7
XS GIS Cut Line= 3
     2377191.746      417061.861     2377153.768      416594.196
     2377174.385      416474.839
#Sta/Elev= 30
       0  421.05       8  420.56    15.9  419.08    23.9  415.38    27.8  415.09
   41.67415.7496    47.7  415.23    55.7  413.41    59.6  413.02   115.3  408.42
   139.2  407.61     167  405.89   250.5  404.15   278.3   402.3  287.52 402.658
   310.2  403.26   314.1  402.98  321.53401.0081   326.1     400     338     401
  345.33402.4807   353.9  403.17   373.8  403.64   433.4  404.16   480.9  406.78
   512.2  409.96   547.4   416.6  568.88419.4357   578.6  421.28   590.3  424.32
#Mann= 7 ,-1 , 0
       0     .12       0   41.67     .06       0  287.52     .12       0
  321.53    .045       0     338     .12       0  345.33     .06       0
  568.88     .12       0
Bank Sta=321.53,338
XS Rating Curve= 0 ,0
Exp/Cntr=0.3,0.1

Type RM Length L Ch R = 1 ,2658.7  ,85.6,90.9,95.4
XS GIS Cut Line= 3
     2377303.508       417046.67     2377649.645      416772.148
     2377763.577      416709.214
#Sta/Elev= 30
       0  413.38    11.9   409.9   23.85409.3012    39.8  408.44   68.11405.4916
   111.4  402.94   175.1   401.8   214.9  400.32   231.2 399.023   238.8   398.4
  244.39397.1555   250.7  395.87   254.7  396.19  259.56 397.222   266.7  399.33
   358.2  399.59     402  400.38   430.1401.7833   449.7  403.22   465.4  405.23
   481.2  408.97     497  413.44   512.8  416.49   516.7  417.62   524.6  420.97
   528.6  421.34   536.4  419.93   540.4  419.99   552.2  424.19   571.9  432.88
#Mann= 7 ,-1 , 0
       0     .12       0   23.85    .016       0   68.11     .06       0
   231.2     .12       0  244.39    .045       0  259.56     .06       0
   430.1     .12       0
#XS Ineff= 2 , 0
                          375.23          401.08
Permanent Ineff=
       F       F
Bank Sta=244.39,259.56
XS Rating Curve= 0 ,0
Exp/Cntr=0.3,0.1

Type RM Length L Ch R = 1 ,2567.9  ,67.4,67.2,67
XS GIS Cut Line= 3
      2377333.89      417072.712     2377745.131      416862.208
     2377813.491      416763.467
#Sta/Elev= 30
       0  413.85   26.18411.2062   34.14 410.532    51.8  409.38    67.7  406.42
   75.17406.1447    83.6  405.87   131.4  402.78  176.13401.6274     223  400.14
     227  399.72   243.8  394.67   246.9  394.02   250.9  393.67   254.9  393.82
   258.8   394.7   270.8  397.47   274.8  398.14   278.8  398.35   378.4  399.42
  413.92400.0823   442.1  400.53     458  403.03   473.6  407.16   489.1  410.82
   512.4   418.6   531.7  425.73   551.1     432   566.6   435.7   582.1  437.69
#Mann= 8 ,-1 , 0
       0     .06       0   26.18     .08       0   34.14     .06       0
   75.17    .016       0  176.13     .06       0   243.8    .045       0
   258.8     .06       0  413.92     .12       0
#XS Ineff= 2 , 0
                           274.3           399.8
Permanent Ineff=
       F       F
Bank Sta=243.8,258.8
XS Rating Curve= 0 ,0
Exp/Cntr=0.3,0.1

Type RM Length L Ch R = 1 ,2500.6  ,136.9,142.4,149
XS GIS Cut Line= 3
     2377361.017      417133.476     2377772.258      416922.972
     2377857.978      416959.865
#Sta/Elev= 30
       0  410.81    47.8  408.62    79.6  406.63    91.6  406.34   103.6  405.27
   115.5  404.67   179.2  402.08  203.21400.2468   211.1  399.28     223  397.22
  233.28394.3915     239  393.34   242.9  393.34  249.31394.4284   258.9  396.46
   286.8  397.41   318.6  400.39   334.5  400.69   346.5  399.65   370.4  400.86
   386.3  400.24   406.2   400.7  420.45401.7425   426.1  401.27   434.1  401.18
   446.1  401.89  470.06402.3385   485.3  403.61   520.3   403.5   555.3  404.48
#Mann= 6 ,-1 , 0
       0     .06       0  203.21     .12       0  233.28    .045       0
  249.31     .12       0  420.45    .016       0  470.06     .12       0
#XS Ineff= 2 , 0
          220.43  398.96  259.44          399.47
Permanent Ineff=
       F       F
Bank Sta=233.28,249.31
XS Rating Curve= 0 ,0
Exp/Cntr=0.3,0.1

Type RM Length L Ch R = 1 ,2358.2  ,192.5,195.2,195.8
XS GIS Cut Line= 3
     2377463.013       417273.45     2377522.692      417177.964
     2377875.339      417100.924
#Sta/Elev= 30
       0  422.27    97.1  413.08   112.6  412.06   132.4  411.56  142.85410.5556
   172.1  404.86     180  401.49     184  399.35     188  396.43   191.9  394.74
   199.9  394.35   202.2393.6469   207.8  392.03   211.8   391.8   215.7  392.83
  216.93393.6589   219.7  395.52   223.7  397.22   227.6  397.52   251.4   396.4
   267.3  396.85   283.2  396.35   291.1  396.83     307  396.16   314.9  396.89
   350.6  397.17     426  401.65   437.9  401.89  460.89 404.029   473.6  406.92
#Mann= 5 ,-1 , 0
       0     .06       0  142.85     .12       0   202.2    .045       0
  216.93     .12       0  460.89    .016       0
#XS Ineff= 2 , 0
                          226.52          397.98
Permanent Ineff=
       F       F
Bank Sta=202.2,216.93
XS Rating Curve= 0 ,0
Exp/Cntr=0.3,0.1

Type RM Length L Ch R = 1 ,2163    ,179.6,178.4,176.3
XS GIS Cut Line= 2
     2377494.046      417366.288     2377898.994      417306.392
#Sta/Elev= 30
       0  422.81    15.9  420.78    47.7  415.35   69.39412.0512    91.4     408
    99.4  407.01   111.3  404.48   115.2  402.99   119.2   400.3   127.2  392.52
   131.2  390.91   135.1   390.7   143.1  391.21     147  392.67     151  394.53
     155  395.83     159  396.12   194.7  393.93   230.5  394.38   242.4   394.2
   258.3  394.86   266.3  394.49   290.1  394.92   329.9   396.4   345.8  397.62
   357.7  399.39   361.7  400.44   369.6  401.04   389.5  403.61   409.4   408.7
#Mann= 4 ,-1 , 0
       0     .06       0   69.39     .12       0   127.2    .045       0
     147     .12       0
#XS Ineff= 2 , 0
                             258          396.21
Permanent Ineff=
       F       F
Bank Sta=127.2,147
XS Rating Curve= 0 ,0
Exp/Cntr=0.3,0.1

Type RM Length L Ch R = 1 ,1984.6  ,270.8,277.2,283
XS GIS Cut Line= 4
     2377511.841      417528.441     2377625.773      417528.441
     2377823.256      417480.698     2377921.997      417476.358
#Sta/Elev= 30
       0  423.78    23.6  421.15    35.4  418.87   53.88414.3559    74.6  408.57
    98.2   400.3   106.1   398.4   121.9  395.85   137.8  394.98   141.8  393.77
  146.81390.0191   149.8  388.65   153.8  388.49   157.8  388.81  163.47389.9781
   173.7  391.38   185.6  394.33   205.6  393.58   221.5  393.89   233.4  393.27
   245.4  393.68   281.2   393.5   297.2  394.68   309.1  394.89     325  396.18
   364.6  403.65   372.4  406.37   384.3  408.28   392.2  411.31   415.9  417.22
#Mann= 4 ,-1 , 0
       0     .06       0   53.88     .12       0  146.81    .045       0
  163.47     .12       0
Bank Sta=146.81,163.47
XS Rating Curve= 0 ,0
Exp/Cntr=0.3,0.1

Type RM Length L Ch R = 1 ,1707.4  ,301,301,298.3
XS GIS Cut Line= 3
     2377503.161      417745.455     2377582.371      417779.092
     2377913.317      417784.517
#Sta/Elev= 30
       0   410.5    27.4  404.02    35.2  401.33      43  397.54    46.9  396.24
    58.7  394.53    67.1393.8292  104.15392.2208     114  392.14   157.8  390.21
   161.8  389.76  164.73388.6698   169.8  387.15   173.8  387.24   181.8  388.67
   189.7  389.61   201.7  389.55   209.7     389   225.6  389.81   237.6  391.43
   245.6  393.52   253.6  394.66   273.5   395.2   285.4  396.44   313.4  398.03
   345.3  401.22   361.2  402.08   369.2  403.66   381.2  404.19     417  407.06
#Mann= 5 ,-1 , 0
       0     .12       0    67.1     .06       0  104.15     .12       0
  164.73    .045       0   181.8     .12       0
Bank Sta=164.73,181.8
XS Rating Curve= 0 ,0
Exp/Cntr=0.3,0.1

Type RM Length L Ch R = 1 ,1406.3  ,465.4,466.8,467.9
XS GIS Cut Line= 4
     2377463.013      418113.294     2377586.711       418052.53
     2377816.746      418043.849     2377928.508      418004.787
#Sta/Elev= 30
       0  412.23    11.8  409.71   27.08409.0951    47.2  408.12    55.1   408.8
    59.1  407.52    66.9  403.11   83.46 397.751    98.4  394.88   133.9  390.18
   157.7  388.52  201.56 386.958   225.1  386.93   229.1  386.54  234.97384.8037
     241   383.5     245  383.56  250.59384.7932   260.8  386.89   276.7  388.91
   304.5  389.32   340.2  391.73     364   392.3   375.9  393.51   399.6  393.92
   423.3  395.59   431.2  396.35     439  397.96   470.6  401.21   486.4   403.7
#Mann= 6 ,-1 , 0
       0     .08       0   27.08     .12       0   83.46     .06       0
  201.56     .12       0  234.97    .045       0  250.59     .12       0
#XS Ineff= 2 , 0
                          280.19          389.28
Permanent Ineff=
       F       F
Bank Sta=234.97,250.59
XS Rating Curve= 0 ,0
Exp/Cntr=0.3,0.1

Type RM Length L Ch R = 1 ,939.5   ,367.1,369.1,370.4
XS GIS Cut Line= 2
     2377514.011      418432.304     2377970.826      418419.283
#Sta/Elev= 30
       0  406.83    23.8  404.23    59.6  401.79    83.4  399.66   103.3  396.04
   119.2  391.94   135.1  388.86     147  387.28     159  386.27   182.8  384.85
   203.9  380.16   206.6  379.05   210.6  378.25   214.6  378.85   218.6  380.37
   222.5  382.37   226.5   383.8   230.5  384.47   242.4  385.35   258.3  385.07
   290.1  385.86     298   386.4     306  386.17   321.9  387.16   361.6  387.67
   377.5  388.92   405.3   394.6   417.3   398.7   445.1  409.92     457  413.99
#Mann= 3 ,-1 , 0
       0     .12       0   203.9    .045       0   218.6     .12       0
Bank Sta=203.9,218.6
XS Rating Curve= 0 ,0
Exp/Cntr=0.3,0.1

Type RM Length L Ch R = 1 ,570.4   ,226.1,217.1,207.2
XS GIS Cut Line= 3
     2377637.709      418713.337     2377935.018      418710.082
     2378010.973       418686.21
#Sta/Elev= 30
       0  396.84    23.8  394.33    31.7  393.75    43.6  392.12    47.6  392.09
    79.3  389.01   142.7  385.94   158.6  385.82   170.5  386.59   182.4  385.25
   194.2  385.21   202.2  384.77     218   382.2     222   380.5     226  376.91
  226.97376.3815   229.9  374.77   233.9  374.39   237.9  374.71  242.55376.2625
   257.7  384.55   261.6  385.88   277.5  386.27   293.4   387.9   301.3  389.62
   309.3  390.96   325.2  394.63   341.1   400.9   349.1  403.57   376.9  413.92
#Mann= 3 ,-1 , 0
       0     .12       0  226.97    .045       0  242.55     .12       0
Bank Sta=226.97,242.55
XS Rating Curve= 0 ,0
Exp/Cntr=0.3,0.1

Type RM Length L Ch R = 1 ,353.3   ,158.3,157.3,156.5
XS GIS Cut Line= 4
     2377686.537      418957.478     2377801.555      418963.988
      2377958.89      418892.373     2378057.631      418877.182
#Sta/Elev= 30
       0  396.92    35.8  392.68    51.6  391.97    59.6  390.79    71.5   389.9
    95.3  388.53   150.6  386.64   174.1  384.84   178.1  384.08     182  382.01
   189.8  375.62   193.8   373.4   197.7  372.44   205.6  372.67  209.99373.3799
   217.4  377.65   221.3  379.39   229.1  381.86   240.9   386.7   244.8  387.39
   264.5  386.97   280.2  387.56   292.1  388.85     304  391.04     312  391.64
     328  393.84     344  397.83     352  400.53     364  404.95     388  414.99
#Mann= 3 ,-1 , 0
       0     .12       0   193.8    .045       0  209.99     .12       0
Bank Sta=193.8,209.99
XS Rating Curve= 0 ,0
Exp/Cntr=0.3,0.1

Type RM Length L Ch R = 1 ,196.1   ,198.1,196.1,193.9
XS GIS Cut Line= 2
     2377759.237      419153.875     2378060.886       418998.71
#Sta/Elev= 30
       0  398.58       8  395.92    23.9  392.25    27.9  391.51    43.9  390.21
    91.8  388.88   127.7  389.69   131.7  389.14   143.7  388.83   151.6  387.87
   155.6  386.99   163.6  382.91   167.6  379.38   171.6  374.14  174.07372.4035
   175.6  371.33   183.6  370.64   187.6  371.48  189.17372.3879   195.6  376.41
   199.5  378.31   219.5  386.21   227.5  388.84   259.4  392.06   271.4  393.61
   283.4  396.01   295.3  399.26   311.3  405.85   323.2  411.42   339.2  416.04
#Mann= 3 ,-1 , 0
       0     .12       0  174.07    .045       0  189.17     .12       0
Bank Sta=174.07,189.17
XS Rating Curve= 0 ,0
Exp/Cntr=0.3,0.1

Chan Stop Cuts=-1
Use User Specified Reach Order=0
Composite Channel Slope=5
